--- BoothsCk.prj (project) ---

Proj Title=BoothsCk
Current Plan=p01
Default Exp/Contr=0,0
English Units
Geom File=g01
Flow File=f01
Plan File=p01
BEGIN DESCRIPTION:
END DESCRIPTION:
DSS Export Rating Curves= 0
DSS Export Rating Curve Sorted= 0
DSS Export Volume Flow Curves= 0
DXF Filename=m:\Didavi\Junko\BoothsCk.
DXF OffsetX= 0
DXF OffsetY= 0
DXF ScaleX= 0
DXF ScaleY= 0

--- BoothsCk.p01 (plan) ---

Plan Title=Floodplain
Program Version=4.00
Geom File=g01
Flow File=f01
K Sum by GR=0
Std Step Tol=0.01
Critical Tol=0.01
Num of Std Step Trials=20
Max Error Tol=0.3
Flow Tol Ratio=0.001
Split Flow NTrial=30
Split Flow Tol=0.02
Split Flow Ratio=0.02
Log Output Level=0
Friction Slope Method=1
Unsteady Friction Slope Method=2
Unsteady Bridges Friction Slope Method=1
Global Log Level=0
CheckData=False
Run HTab=0
Run UNet=0
Run PostProcess=0
UNET Theta=0
UNET Theta Warmup=0
UNET ZTol=0
UNET ZSATol=0
UNET MxIter=0
UNET MaxInSteps=0
UNET DtIC=0
UNET DtMin=0
UNET MaxCRTS=0
UNET WFStab=0
UNET SFStab=0
UNET WFX=0
UNET SFX=0
UNET DSS MLevel=0
UNET DZMax Abort=0
UNET Convert EG Bridges=0
UNET Use Existing IB Tables=0
UNET Froude Limit=0
UNET Froude Power=0
Write IC File=0
Echo Input=False
Echo Output=False
Write Detailed=0

--- BoothsCk.f01 (steady flow) ---

Flow Title=NFF Regression Equation
Program Version=4.10
Number of Profiles= 1
Profile Names=P100yr
River Rch & RM=BoothsCk,Main            ,42296.3
     874
River Rch & RM=BoothsCk,Main            ,39116.6
    1506
River Rch & RM=BoothsCk,Main            ,38727
    1644
River Rch & RM=BoothsCk,Main            ,36670.4
    1752
River Rch & RM=BoothsCk,Main            ,33571.3
    1798
River Rch & RM=BoothsCk,Main            ,33179.7
    1898
River Rch & RM=BoothsCk,Main            ,32352.4
    1951
River Rch & RM=BoothsCk,Main            ,27616.4
    2063
River Rch & RM=BoothsCk,Main            ,25481.5
    2431
River Rch & RM=BoothsCk,Main            ,22963.2
    3275
River Rch & RM=BoothsCk,Main            ,18283.1
    3420
River Rch & RM=BoothsCk,Main            ,8885.4
    3681
River Rch & RM=BoothsCk,Main            ,6181.7
    3722
River Rch & RM=BoothsCk,Main            ,5397.1
    4054
River Rch & RM=BoothsCk,Main            ,4503.5
    4059
Boundary for River Rch & Prof#=BoothsCk,Main            , 1
Up Type= 0
Dn Type= 3
Dn Slope=0.007218
DSS Import GetInterval= 0
DSS Import GetPeak= 0
DSS Import FillOption= 0

--- BoothsCk.g01 (geometry) ---

Geom Title=USGS 10m DEM
Program Version=4.10

River Reach=BoothsCk        ,Main
Reach XY= 30
     1841138.278      364460.052     1840674.718      364991.737
     1839586.055       365314.66     1839246.185      365962.866
     1837691.095      366489.998      1837225.85      366978.514
     1837731.903      369350.776     1836740.116       370953.25
      1837004.02         372035.      1836184.74      374036.785
     1835730.118      374785.157     1833783.558      375495.925
     1833396.978      376025.924     1833990.653      377871.042
     1832914.304       379208.21     1833028.237      379913.288
      1832681.05      380351.221     1832581.931      381784.937
     1833098.053       382835.95      1832150.48      383361.524
     1832069.456      383989.863     1833035.394      384835.211
      1832566.47      385794.668     1832880.436      385975.621
     1833017.367      388850.614     1835079.825      391566.582
     1834868.019      391983.248     1835203.957      392863.804
     1834387.984      394491.235     1834065.783       396842.18

Type RM Length L Ch R = 1 ,42296.3 ,277.8,285.2,292.2
XS GIS Cut Line= 2
     1840841.408      364307.177     1841352.057      364583.977
#Sta/Elev= 30
       0  1447.4    29.5 1438.61    39.4 1435.09    88.6 1412.64   108.3 1404.81
   118.1 1400.46     128 1399.16   137.8  1396.6   147.7 1393.25   177.2 1381.05
   196.9  1373.7   226.4 1364.58     256 1356.48   265.8 1352.74   285.5 1344.07
     315 1329.37   324.9 1325.25   325.4 1325.27   334.7 1325.55   340.51326.425
   364.3  1331.2   374.1 1334.12     384 1338.33   413.5 1354.32   423.3 1359.06
   433.2 1361.97   462.7 1369.56   472.6 1371.18   551.3 1379.89   580.8 1383.62
#Mann= 3 , 0 , 0
       0      .1       0   325.4    .045       0   340.5      .1       0
Bank Sta=325.4,340.5
XS Rating Curve= 0 ,0
Exp/Cntr=0.3,0.1

Type RM Length L Ch R = 1 ,42011   ,285.7,285.5,285.4
XS GIS Cut Line= 2
     1840869.111      364534.193     1841181.688      364892.579
#Sta/Elev= 30
       0 1382.86     9.9 1373.34    19.8 1365.05    39.6 1350.86    49.5 1344.35
    59.4 1338.49    69.4 1333.54    79.3 1329.41    89.2 1327.86   138.7 1322.32
   148.6 1319.92   154.11318.052   158.5 1316.56   168.4 1316.55   169.61316.682
   188.2 1318.58   198.1 1318.89     208 1318.09     218 1318.77   257.6 1323.04
   277.4 1323.29   287.3 1324.79   297.2 1327.87   307.1  1332.5   326.9 1344.38
   346.8 1355.66   356.7 1359.62   406.2 1369.25   435.9 1377.92   475.6 1388.12
#Mann= 3 , 0 , 0
       0      .1       0   154.1    .045       0   169.6      .1       0
Bank Sta=154.1,169.6
XS Rating Curve= 0 ,0
Exp/Cntr=0.3,0.1

Type RM Length L Ch R = 1 ,41725.5 ,344.7,347.9,351
XS GIS Cut Line= 2
     1840623.451       364678.29     1840936.028      365036.676
#Sta/Elev= 30
       0 1387.38     9.9 1383.41    19.8 1378.25    39.6 1376.45     109 1350.45
   118.9 1347.56   138.7  1343.3   168.4 1334.81   188.2 1327.68   198.1 1323.24
     208 1316.97     218 1312.08   227.9 1309.39   254.7 1304.75   257.6 1304.24
   267.5 1305.32   269.7 1306.15   277.4 1309.04   287.3 1311.49   307.1 1310.96
     317 1311.55   336.8 1317.05   346.8  1321.3   356.7 1327.08   366.6  1333.8
   376.5 1336.42   386.4 1337.92   406.2 1347.82   455.7 1367.01   475.6 1373.93
#Mann= 3 , 0 , 0
       0      .1       0   254.7    .045       0   269.7      .1       0
Bank Sta=254.7,269.7
XS Rating Curve= 0 ,0
Exp/Cntr=0.3,0.1

Type RM Length L Ch R = 1 ,41377.6 ,525.4,537.1,548.9
XS GIS Cut Line= 2
     1840389.404       364814.24     1840634.938       365217.98
#Sta/Elev= 30
       0 1383.32     9.8 1377.72    39.4 1363.57    49.2 1356.85    59.1 1353.79
    68.9 1353.74    78.8  1351.2    98.4 1343.48   118.1 1334.89     128 1329.09
   137.8  1326.2   167.4 1308.55   177.2  1302.2     187 1296.67   196.9 1292.93
     1991292.561   206.7 1291.19   215.61291.452   236.3 1293.73   265.8 1295.34
   275.6 1297.25   295.3 1302.69   305.2 1306.37   334.7  1319.2   344.6 1321.49
   364.2    1324   403.6 1325.06     443 1327.84   452.8 1329.13   472.5 1333.36
#Mann= 3 , 0 , 0
       0      .1       0     199    .045       0   215.6      .1       0
Bank Sta=199,215.6
XS Rating Curve= 0 ,0
Exp/Cntr=0.3,0.1

Type RM Length L Ch R = 1 ,40840.5 ,194.9,190.3,186
XS GIS Cut Line= 2
     1840057.154      365007.036      1840084.64      365389.988
#Sta/Elev= 30
       0 1316.33     9.8 1315.84    19.7 1314.37    39.4 1309.05    49.2 1306.73
    78.8 1300.05    88.6 1298.71    98.4 1295.85   108.3    1287   118.1 1278.97
     128 1272.87   137.8 1271.39   147.7 1269.14   150.91268.015   157.5 1265.69
   167.4 1266.87     187 1272.11   196.9 1274.08   216.6 1277.04   226.4  1278.3
   236.3  1279.1   265.8    1280   275.6 1280.81   295.3 1283.04   305.2 1285.03
   324.9  1290.5   334.7 1291.96   364.2  1293.5   374.1 1293.82   383.9 1293.78
#Mann= 3 , 0 , 0
       0      .1       0   150.9    .045       0   167.4      .1       0
Bank Sta=150.9,167.4
XS Rating Curve= 0 ,0
Exp/Cntr=0.3,0.1

Type RM Length L Ch R = 1 ,40650.2 ,300.8,298.4,295.3
XS GIS Cut Line= 2
     1839814.976      364963.022     1839952.187      365438.001
#Sta/Elev= 30
       0 1312.29    49.4 1304.37    79.1  1298.6    98.9 1297.05   118.7 1294.27
   138.4 1289.68   148.3 1286.72   158.2 1283.02   168.1 1280.94     178 1277.94
   187.9  1273.3   197.8 1271.48   217.5  1265.7   247.2 1259.99   281.71255.257
   286.8  1254.4   296.6 1253.84   298.1  1254.2   306.5 1256.24   326.3 1263.49
   346.1 1269.42   365.9 1270.95   385.6 1269.97   405.4 1269.74   415.3 1271.38
   425.2 1273.91   435.1 1277.26     445 1279.17   474.6 1281.36   494.4 1281.39
#Mann= 3 , 0 , 0
       0      .1       0   281.7    .045       0   298.1      .1       0
Bank Sta=281.7,298.1
XS Rating Curve= 0 ,0
Exp/Cntr=0.3,0.1

Type RM Length L Ch R = 1 ,40351.9 ,415.3,393.7,372.9
XS GIS Cut Line= 2
      1839492.33      364994.073     1839743.934       365617.27
#Sta/Elev= 30
       0 1294.49    69.2 1286.81   118.6 1283.18   148.2 1280.36     168 1278.13
   177.9 1276.19   187.8 1275.44   207.6 1275.99   227.3 1274.44   247.1 1271.86
   276.7 1263.19   296.5 1255.02   306.4  1252.8   324.8 1244.35     336 1241.47
   345.9 1244.64   355.8 1247.56   395.3 1254.98   405.2 1255.61   415.1 1255.37
   444.8 1253.21   454.6 1252.98   464.5 1253.66   474.4  1255.2   513.9 1256.72
   563.4 1260.79   573.2 1261.11   602.9 1260.42   632.5 1261.84   672.1 1267.92
#Mann= 3 , 0 , 0
       0      .1       0   324.8    .045       0   345.9      .1       0
Bank Sta=324.8,345.9
XS Rating Curve= 0 ,0
Exp/Cntr=0.3,0.1

Type RM Length L Ch R = 1 ,39958.2 ,814.4,841.5,867
XS GIS Cut Line= 3
       1839115.2      365270.272     1839253.516      365550.171
     1839753.992      365685.224
#Sta/Elev= 30
       0 1264.69    29.3 1261.04    58.5 1255.04      78 1249.89    97.6 1246.79
   117.1 1241.54   126.8 1237.11   136.6 1236.34   146.4 1237.43   204.9  1239.1
   234.2 1237.08   292.7  1236.2   342.1 1238.99     362 1238.98     372  1237.2
     382 1233.39     392 1230.63   401.9 1230.29   411.9 1231.98   461.7 1235.72
   501.6 1235.99   511.6    1238   551.5 1240.72   561.4 1242.07   581.4 1246.81
   591.3 1247.85   720.9 1258.52   730.9 1259.72   800.7 1273.15   830.6 1277.17
#Mann= 3 , 0 , 0
       0      .1       0     382    .045       0   411.9      .1       0
Bank Sta=382,411.9
XS Rating Curve= 0 ,0
Exp/Cntr=0.3,0.1

Type RM Length L Ch R = 1 ,39116.6 ,400,389.6,379.2
XS GIS Cut Line= 2
     1838803.919      365699.242     1838966.027      366462.551
#Sta/Elev= 30
       0  1275.7    59.3 1253.38      79 1244.53    88.9 1243.69    98.8 1241.11
   167.9 1219.67   187.7  1217.1   227.2 1216.97   237.1 1215.83   257.3 1210.79
   266.7 1209.94   276.6 1210.67   306.2    1216   316.1 1216.86   355.6 1216.87
   375.4 1218.26   385.2 1220.23   395.1 1223.27   414.9 1231.02   464.2 1242.17
     484 1245.53   503.8 1246.22   523.5 1253.05   602.5 1277.09     642 1285.89
   721.1  1301.4   740.8 1306.51   750.7 1306.94   760.6 1310.67   780.3 1315.95
#Mann= 3 , 0 , 0
       0      .1       0   257.3    .045       0   276.6      .1       0
Bank Sta=257.3,276.6
XS Rating Curve= 0 ,0
Exp/Cntr=0.3,0.1

Type RM Length L Ch R = 1 ,38727   ,421.5,424.9,428.6
XS GIS Cut Line= 2
     1838308.376      365863.172     1838648.754      366293.339
#Sta/Elev= 30
       0  1322.4      20 1315.22    69.8 1295.99    79.8 1293.18    89.8 1292.03
    99.7 1289.24   119.7 1282.77   129.7  1280.9   149.6 1273.29   159.6  1269.1
   189.5 1253.96   199.5 1248.52   209.4 1241.93   229.4 1230.33   249.3 1221.64
   259.3 1217.68   269.3 1214.38   289.2 1209.03   299.2 1205.73   301.71205.345
   309.2  1204.2   316.91204.707   339.1 1207.64     369 1209.82   398.9 1211.25
   438.8  1215.7   468.8 1220.44   498.7 1225.78   528.6 1231.57   548.5 1236.04
#Mann= 3 , 0 , 0
       0      .1       0   301.7    .045       0   316.9      .1       0
Bank Sta=301.7,316.9
XS Rating Curve= 0 ,0
Exp/Cntr=0.3,0.1

Type RM Length L Ch R = 1 ,38302.1 ,550,549.5,547.7
XS GIS Cut Line= 2
     1837991.747      366076.618     1838301.989      366575.068
#Sta/Elev= 30
       0 1283.04      10 1279.18   119.4 1246.74   139.3 1239.06   179.1  1220.8
   189.1 1216.98     199 1214.78     209 1211.44   218.9 1208.93   228.9 1206.89
   238.8 1205.59   278.6 1202.81   288.6 1202.59   298.5 1203.39   328.4 1203.77
   338.3 1203.44   349.71201.707   358.2 1201.26   366.61201.328     408 1202.09
   427.9 1209.12   467.7 1221.39   487.6 1228.01   497.6 1232.26   507.5  1237.2
   537.4 1247.94   547.3 1252.44   557.3 1255.58   577.2 1257.24   587.1 1263.29
#Mann= 3 , 0 , 0
       0      .1       0   349.7    .045       0   366.6      .1       0
Bank Sta=349.7,366.6
XS Rating Curve= 0 ,0
Exp/Cntr=0.3,0.1

Type RM Length L Ch R = 1 ,37752.7 ,349.4,343,336.9
XS GIS Cut Line= 2
     1837571.413      366280.499     1837935.245      366822.753
#Sta/Elev= 30
       0 1288.56    29.7 1271.42    49.5 1264.04      89 1246.33    98.9 1243.24
   118.7  1239.8   128.6 1236.87   158.3 1224.28   168.2  1220.9   197.9 1213.42
   207.8 1208.48   217.7 1201.98   227.6 1194.18   236.21190.345   237.5 1189.76
   251.41190.313   267.1 1192.57   316.6 1193.86   366.1 1197.31   395.8 1197.06
   405.6 1197.86   415.6 1199.74   445.2 1208.11   544.2  1243.2     564 1248.03
   583.8 1248.18   603.5 1255.32   623.3 1261.03   643.1 1262.91     653 1265.54
#Mann= 3 , 0 , 0
       0      .1       0   236.2    .045       0   251.4      .1       0
Bank Sta=236.2,251.4
XS Rating Curve= 0 ,0
Exp/Cntr=0.3,0.1

Type RM Length L Ch R = 1 ,37409.7 ,357.4,352.8,348.2
XS GIS Cut Line= 2
     1837255.767      366543.561     1837711.628      366934.911
#Sta/Elev= 30
       0 1284.68    19.7 1278.64    29.6 1274.69    68.9 1256.68    78.8 1252.64
    88.6 1248.11    98.5 1244.28   108.3  1243.2   118.2  1240.3   137.9 1232.18
   157.6 1226.91   177.3 1220.78   226.5 1202.64   256.1 1189.86   263.8 1186.21
   265.9 1185.21   275.8 1183.77   285.6 1184.95   305.3  1189.3   315.2 1190.32
     325 1190.91   374.3 1191.29   384.1  1192.3   413.7 1197.64   502.3  1222.6
   551.6    1238   571.2 1245.03   581.1  1247.1     591 1247.72   600.8 1251.24
#Mann= 3 , 0 , 0
       0      .1       0   263.8    .045       0   285.6      .1       0
Bank Sta=263.8,285.6
XS Rating Curve= 0 ,0
Exp/Cntr=0.3,0.1

Type RM Length L Ch R = 1 ,37056.9 ,401.6,386.5,371.1
XS GIS Cut Line= 2
     1837012.518      366863.006      1837552.56      367163.868
#Sta/Elev= 30
       0 1200.22    29.9 1199.18    69.8 1198.57   109.7 1197.46   159.5 1199.93
   169.5 1200.01   179.5 1199.46   189.4 1197.76   199.4 1194.86   209.4 1190.64
   219.4 1185.89   229.3 1182.47   235.1 1181.44   239.3  1180.7   250.1 1180.81
   269.2  1182.6   289.2 1182.73   319.1 1181.64     349 1182.58   408.8 1181.33
   418.8 1182.54   438.7 1188.44   498.5 1209.38   548.4 1224.61   568.3 1232.15
   578.3 1233.04   588.3 1233.25   598.2 1239.54   608.2 1245.13   618.2 1249.02
#Mann= 3 , 0 , 0
       0      .1       0   235.1    .045       0   250.1      .1       0
Bank Sta=235.1,250.1
XS Rating Curve= 0 ,0
Exp/Cntr=0.3,0.1

Type RM Length L Ch R = 1 ,36670.4 ,331.6,339.1,346.2
XS GIS Cut Line= 2
     1836996.441      367375.091      1837560.88      367281.138
#Sta/Elev= 30
       0 1223.95    19.7 1217.48    69.1 1202.62    78.9 1199.91    88.8 1197.94
   108.5 1195.46     217 1186.27   226.9 1185.11   256.5 1178.38   286.1 1178.02
   305.8  1176.7   315.7 1175.79   352.3 1170.01   355.2 1169.58     365 1169.61
   367.41170.059   374.9 1171.45   404.5 1180.68   414.4 1184.91   424.2 1190.34
   434.1 1196.82   453.8 1212.47   463.7 1217.23   473.6 1218.98   483.4 1219.71
   493.3 1224.11   503.2 1229.31   532.7 1241.15   552.5 1249.64   572.2 1259.36
#Mann= 3 , 0 , 0
       0      .1       0   352.3    .045       0   367.4      .1       0
Bank Sta=352.3,367.4
XS Rating Curve= 0 ,0
Exp/Cntr=0.3,0.1

Type RM Length L Ch R = 1 ,36331.3 ,630.8,616,601.2
XS GIS Cut Line= 2
     1836986.639      367593.542     1837700.933      367707.663
#Sta/Elev= 30
       0 1224.11    19.8 1212.29    39.6 1204.21    79.3  1194.6     109 1182.91
   118.9  1180.6   138.7 1178.38   168.4 1176.62   198.2 1172.18   247.7 1173.25
   317.1 1172.04     327 1170.82   346.8    1166   356.7 1164.97   376.5  1165.7
   396.4 1169.56   406.3 1172.27   426.1 1180.13     436 1181.33   445.9 1180.89
   465.7 1191.96   505.4 1203.37   515.3 1206.69   535.1 1214.88   554.9 1219.37
   574.7  1227.3   604.4 1237.74   663.9 1261.75   703.5 1274.62   723.4  1278.3
#Mann= 3 , 0 , 0
       0      .1       0   346.8    .045       0   376.5      .1       0
Bank Sta=346.8,376.5
XS Rating Curve= 0 ,0
Exp/Cntr=0.3,0.1

Type RM Length L Ch R = 1 ,35715.3 ,668.2,675.8,683.1
XS GIS Cut Line= 2
     1837111.639      368437.292     1837851.222      368046.667
#Sta/Elev= 30
       0 1243.84    19.9 1239.02    69.7 1220.06   109.5 1203.12   149.4 1183.96
   199.1 1172.37     239 1167.76   268.8 1159.77   298.7 1155.83   328.6 1156.11
   388.3 1159.35   408.2 1158.96   418.2  1156.7   428.2 1153.95   448.1 1155.12
     458 1157.02     478 1155.92   507.8 1157.32   537.7 1157.23   547.6 1158.07
   557.6  1160.7   567.6 1163.93   607.4 1183.18   627.3 1190.98   657.2 1206.44
     707 1228.64   726.9 1235.17   796.6 1254.57   816.5 1258.04   836.4 1264.39
#Mann= 3 , 0 , 0
       0      .1       0   418.2    .045       0   448.1      .1       0
Bank Sta=418.2,448.1
XS Rating Curve= 0 ,0
Exp/Cntr=0.3,0.1

Type RM Length L Ch R = 1 ,35039.5 ,331.5,332,332.5
XS GIS Cut Line= 2
     1837379.673      368846.246     1837991.625      368752.961
#Sta/Elev= 30
       0 1238.29    39.9 1223.77    59.9 1214.99    69.9 1212.68    89.9 1202.65
   109.8 1190.16   139.8 1172.84   149.8 1167.66   169.7 1155.46   179.7 1150.89
   189.7 1147.73   219.6 1146.39   229.6 1144.67   239.6 1143.91   259.6 1144.84
   309.5 1145.21   348.21143.663   359.4 1143.62   363.51144.081   379.4 1146.33
   399.4 1148.36   419.3 1148.01   429.3 1148.91   459.3 1158.68   489.2 1162.83
   529.2 1171.55   549.1 1173.13   569.1 1178.36     599 1182.21     619 1186.49
#Mann= 3 , 0 , 0
       0      .1       0   348.2    .045       0   363.5      .1       0
Bank Sta=348.2,363.5
XS Rating Curve= 0 ,0
Exp/Cntr=0.3,0.1

Type RM Length L Ch R = 1 ,34707.5 ,484.6,490.8,496.7
XS GIS Cut Line= 2
     1837370.136      369155.298     1838055.364      369062.381
#Sta/Elev= 30
       0 1247.77    49.4  1231.1    98.8 1216.05   138.3 1205.59   167.9 1193.86
   187.7 1171.67   197.6 1165.52   207.4 1157.49   217.3 1147.36   227.2 1140.08
   237.1 1137.56     247 1137.23   276.6 1138.82   316.1 1138.63     326 1137.36
   335.9  1136.6   347.31137.532   365.5 1139.89   385.3 1138.53   424.8 1138.73
   444.5 1141.31     484 1143.62   503.8 1147.46   523.6 1148.69     573  1154.8
   602.6 1161.71   612.5 1161.61   642.1 1168.72   661.9 1175.14   691.5 1187.13
#Mann= 3 , 0 , 0
       0      .1       0     326    .045       0   347.3      .1       0
Bank Sta=326,347.3
XS Rating Curve= 0 ,0
Exp/Cntr=0.3,0.1

Type RM Length L Ch R = 1 ,34216.7 ,630.7,645.4,659.9
XS GIS Cut Line= 2
     1837305.749      369517.031     1838052.224      369610.295
#Sta/Elev= 30
       0 1192.49    59.4  1177.9    89.1 1168.38   118.8 1157.31   128.7 1154.06
   148.5 1148.29   178.2 1140.46   188.1 1138.54   207.9 1136.79   227.7 1138.11
   267.3 1136.05   277.2 1135.28     287 1133.75     297 1131.52   316.8 1129.79
   326.6 1128.02   346.4 1128.66   356.3 1130.46   376.1 1131.15   415.7 1133.87
   465.2  1134.3     584 1133.47   633.5 1134.29   653.3 1135.97   673.1 1138.21
     683 1140.17   692.9 1143.17   702.8  1146.5   722.6 1154.66   752.3 1168.88
#Mann= 3 , 0 , 0
       0      .1       0   316.8    .045       0   356.3      .1       0
Bank Sta=316.8,356.3
XS Rating Curve= 0 ,0
Exp/Cntr=0.3,0.1

Type RM Length L Ch R = 1 ,33571.3 ,388.8,391.7,394.5
XS GIS Cut Line= 2
        1837151.      369853.437     1837614.149      370273.482
#Sta/Elev= 30
       0 1134.54     9.9 1133.78    29.8 1126.25    39.7 1124.19    49.6 1123.18
    89.3 1121.75   148.9 1121.78   178.6 1119.43   238.2 1118.83     268 1119.26
   277.9 1118.27   287.8 1115.56   297.7 1114.45   307.7 1114.52   317.6 1116.04
   337.4 1124.61   347.4 1129.46   357.3 1131.39   367.2 1131.44   387.1 1130.72
   466.5 1132.93   516.1 1133.57     526  1133.6   535.9 1133.05   545.9 1132.07
   555.8 1132.14   565.7 1134.01   575.6 1137.36   595.5  1145.7   625.3 1156.63
#Mann= 3 , 0 , 0
       0     .08       0   287.8    .045       0   317.6      .1       0
Bank Sta=287.8,317.6
XS Rating Curve= 0 ,0
Exp/Cntr=0.3,0.1

Type RM Length L Ch R = 1 ,33179.7 ,271.8,262.9,253.8
XS GIS Cut Line= 2
     1836933.715      370135.332     1837286.353      370531.321
#Sta/Elev= 30
       0  1139.3     9.8 1138.57    19.6 1136.94    29.5 1136.31    39.3 1136.37
    58.9 1134.78    68.7 1133.74    88.4 1130.03     108 1128.11   117.8 1124.98
   137.5 1114.67   147.3 1112.31   235.7 1111.44   245.5 1109.74   255.3 1106.52
   265.1 1105.36   274.9 1105.31   284.8 1106.49   294.6 1109.37   314.2  1116.3
     324 1121.02   333.9 1129.05   343.7 1141.18   353.5 1145.13   392.8  1156.5
   402.6 1159.01   422.2 1163.78   461.5 1172.25     491 1179.78   530.2 1191.68
#Mann= 3 , 0 , 0
       0      .1       0   255.3    .045       0   284.8      .1       0
Bank Sta=255.3,284.8
XS Rating Curve= 0 ,0
Exp/Cntr=0.3,0.1

Type RM Length L Ch R = 1 ,32916.8 ,301.9,301.9,301.9
XS GIS Cut Line= 2
     1836677.717      370401.585      1837173.04      370643.645
#Sta/Elev= 30
       0  1145.6    78.8 1134.68    88.6  1133.6   108.3 1132.71   118.1 1131.77
   137.8 1128.51   147.7 1127.76   167.4 1127.82   196.9  1126.6   216.6 1125.25
   226.4 1123.64   246.1 1115.93     256 1114.62   265.8 1111.35   275.6 1107.05
   285.5 1103.85   295.3 1101.03     3001100.472   305.2 1099.85   324.9 1100.48
   334.7 1103.01   344.6 1106.25   354.4 1111.83   374.1 1126.03     384 1131.33
   413.5  1143.2   452.9 1155.83   492.2  1165.3   511.9 1169.52   551.3 1180.42
#Mann= 3 , 0 , 0
       0      .1       0     300    .045       0   324.9      .1       0
Bank Sta=300,324.9
XS Rating Curve= 0 ,0
Exp/Cntr=0.3,0.1

Type RM Length L Ch R = 1 ,32614.9 ,283.6,262.5,241.3
XS GIS Cut Line= 2
     1836519.979       370660.26     1837034.859      370911.878
#Sta/Elev= 30
       0 1164.91    29.6 1156.75    59.3  1146.8      79 1140.96    98.8 1135.66
   128.4 1128.48   148.2 1125.22     168 1122.75   197.6 1120.51   207.5 1119.36
   227.2 1118.66   266.8 1113.85   276.7 1111.32   306.3  1099.1   316.2 1095.39
   326.1  1093.8   335.7 1093.78   345.8  1094.7   355.7 1097.64   375.5 1105.97
   395.2 1107.38     415  1108.3   424.9 1109.54   434.8 1112.06   454.5 1118.86
   464.4 1121.87   484.2 1127.24     494 1129.59   543.4 1139.93   573.1 1145.41
#Mann= 3 , 0 , 0
       0      .1       0   316.2    .045       0   345.8      .1       0
Bank Sta=316.2,345.8
XS Rating Curve= 0 ,0
Exp/Cntr=0.3,0.1

Type RM Length L Ch R = 1 ,32352.4 ,462.4,467.2,472
XS GIS Cut Line= 2
     1836514.498      371161.344     1836943.427      370947.321
#Sta/Elev= 30
       0 1166.51      40 1153.99    69.9 1146.05    79.9 1143.03    89.9 1141.91
   109.8 1137.18   129.8 1133.13   139.8 1130.04   149.8 1125.45   169.8 1122.14
   189.8 1111.13   209.7 1101.66   219.7  1097.6   239.7 1091.76   244.31090.849
   249.7 1089.78   255.1 1089.77   259.6 1089.77   270.1 1090.52   279.6    1094
   289.6 1098.55   299.6  1100.1   329.6 1100.67   339.6 1101.88   349.5 1102.64
   369.5 1103.66   429.4  1105.1   439.4 1106.31   459.4 1110.86   479.4 1117.24
#Mann= 3 , 0 , 0
       0      .1       0   244.3    .045       0   270.1      .1       0
Bank Sta=244.3,270.1
XS Rating Curve= 0 ,0
Exp/Cntr=0.3,0.1

Type RM Length L Ch R = 1 ,31885.2 ,562.6,575.6,588.6
XS GIS Cut Line= 2
     1836756.034      371504.814     1837219.256      371385.277
#Sta/Elev= 30
       0 1101.99    39.9 1099.86    49.8  1097.8    69.8 1096.74    79.7 1095.34
    89.7 1093.06    99.7 1091.61   119.6 1090.47   159.5 1089.95   179.4  1089.2
   189.4  1088.1   199.3 1086.66   209.3 1084.38   219.3 1083.97   239.2 1084.14
   249.2 1085.38   269.1 1088.54     309 1090.74   328.9 1092.75   338.9 1094.52
   358.8 1098.93   368.8 1101.87   398.7 1111.42   418.6 1117.38   428.6 1119.86
   438.5 1121.45   448.5 1122.74   458.5 1124.84   468.4 1127.97   478.4 1131.52
#Mann= 3 , 0 , 0
       0      .1       0   209.3    .045       0   239.2      .1       0
Bank Sta=209.3,239.2
XS Rating Curve= 0 ,0
Exp/Cntr=0.3,0.1

Type RM Length L Ch R = 1 ,31309.6 ,405.1,412.4,419.7
XS GIS Cut Line= 2
     1836773.361      371944.132     1837253.351      372103.665
#Sta/Elev= 30
       0 1078.38    39.7 1076.83    99.2 1073.72   128.9  1072.6   148.8 1070.64
   158.7 1070.01   198.4 1068.72   208.3 1067.89   218.2 1065.15   228.1 1060.98
     248 1060.61   257.9 1060.97   267.8 1066.12   277.7  1073.8   297.5 1087.43
   307.4 1095.69   327.3 1106.38   337.2 1113.75   347.1 1121.58     367 1138.56
   376.9 1146.07   406.6 1167.43   416.6 1172.58   436.4 1181.82   446.3 1187.53
   456.2 1194.51   466.1 1201.11     476 1207.19   495.9 1218.18   505.8 1223.34
#Mann= 3 , 0 , 0
       0      .1       0   228.1    .045       0   257.9      .1       0
Bank Sta=228.1,257.9
XS Rating Curve= 0 ,0
Exp/Cntr=0.3,0.1

Type RM Length L Ch R = 1 ,30897.2 ,598.9,602.3,605.8
XS GIS Cut Line= 2
      1836619.44      372234.511     1837044.211      372554.329
#Sta/Elev= 30
       0 1067.96    98.5 1064.33   137.8 1063.46   157.5 1063.71   167.4 1063.31
   177.2 1061.62   187.1 1060.94   196.9 1061.45   206.8 1058.86   216.6 1056.89
   226.5 1056.24   246.2 1055.77   255.61054.919   265.8  1054.4   275.7  1054.4
   285.6 1054.65   295.4 1059.31   305.2 1067.47   315.1 1074.74   324.9 1081.81
   344.6 1094.95   354.5  1100.9   364.3 1107.24   374.2 1112.49     384 1116.32
   393.9 1118.51   403.7 1119.78   443.1 1123.41   452.9 1124.07   531.7 1127.08
#Mann= 3 , 0 , 0
       0      .1       0   255.6    .045       0   285.6      .1       0
Bank Sta=255.6,285.6
XS Rating Curve= 0 ,0
Exp/Cntr=0.3,0.1

Type RM Length L Ch R = 1 ,30294.9 ,609.6,596.8,584.1
XS GIS Cut Line= 2
     1836188.301      372603.603     1836726.022       373069.65
#Sta/Elev= 30
       0 1067.33    59.3 1064.11   118.6 1058.25   158.1 1055.92     168 1056.23
   266.8 1053.38   365.7 1052.23   375.6 1051.34   385.4 1049.62   395.3 1048.99
   405.2 1049.14   415.1 1047.85     425 1046.55   444.7 1046.38   454.6 1046.54
   484.3 1048.43   494.2 1050.58     504 1056.58   523.8 1070.95   543.6 1087.35
   553.4 1096.52   563.3 1100.28   573.2 1104.82   583.1 1113.21     593 1117.42
   632.5 1129.53   662.2 1137.55   681.9 1143.92   691.8 1146.21   711.6 1152.21
#Mann= 3 , 0 , 0
       0     .08       0   415.1    .045       0   454.6      .1       0
Bank Sta=415.1,454.6
XS Rating Curve= 0 ,0
Exp/Cntr=0.3,0.1

Type RM Length L Ch R = 1 ,29698.1 ,850.7,848,844.7
XS GIS Cut Line= 4
     1835828.863      373112.347     1836113.823      373261.865
     1836166.123      373396.351     1836579.269      373489.009
#Sta/Elev= 30
       0 1092.76    19.5 1083.15    29.2 1080.08    48.8 1075.88    87.8 1069.68
   136.5 1066.26   165.8 1059.82   185.3 1056.79     195 1054.21   224.3 1049.42
   253.5 1047.23   292.6 1045.81   360.3  1046.7   505.5 1045.35   515.3 1044.71
     535 1040.65   544.9 1039.98   564.6 1040.24     604 1041.61   613.8 1042.79
   623.6 1046.76   633.5 1052.32   653.2 1064.74   672.9 1081.68   682.7 1088.45
   712.3 1100.08   771.4 1116.56   800.9 1125.41   869.8 1148.27   889.5 1155.66
#Mann= 3 , 0 , 0
       0      .1       0     535    .045       0   564.6      .1       0
Bank Sta=535,564.6
XS Rating Curve= 0 ,0
Exp/Cntr=0.3,0.1

Type RM Length L Ch R = 1 ,28850.1 ,465.7,471.5,477.4
XS GIS Cut Line= 2
     1835638.417      374057.294     1836444.903      374149.947
#Sta/Elev= 30
       0 1131.13     9.9 1124.65    19.8 1120.25    39.6 1116.78    59.4 1105.72
    89.1 1105.91   108.9  1095.8   118.8 1091.75   148.5 1082.48   227.7 1062.05
   247.5 1057.78   267.3 1049.59   287.1 1042.77     297 1040.57   326.7 1038.87
   336.6 1034.73   346.5 1031.71   356.4 1031.54   376.2 1032.93   514.8 1035.32
   524.7 1035.83   554.4 1041.27   584.1 1052.25   613.8 1056.87   623.7 1060.37
   643.5 1071.65   683.1 1086.81   722.7 1105.68   782.1 1129.34   811.8 1142.96
#Mann= 3 , 0 , 0
       0      .1       0   336.6    .045       0   376.2      .1       0
Bank Sta=336.6,376.2
XS Rating Curve= 0 ,0
Exp/Cntr=0.3,0.1

Type RM Length L Ch R = 1 ,28378.5 ,741,762.1,782.8
XS GIS Cut Line= 2
     1835577.206      374428.641     1836325.459      374708.128
#Sta/Elev= 30
       0 1077.35      10 1075.73      30 1068.85    59.9 1067.78   129.8 1052.46
   179.7 1045.84   199.7 1041.15   229.6  1030.5   258.9 1026.15   269.6 1025.75
   279.6 1026.29   289.6 1027.81   349.4 1029.02   389.4 1031.85   479.2 1035.14
   509.2 1037.97   519.2 1041.91   569.1 1069.95   599.1 1089.59     609 1095.27
     629 1098.22     659 1099.96     669 1103.01   688.9 1113.02   708.9 1127.83
   718.9 1132.26   728.9 1133.75   738.8 1136.75   778.8 1149.41   798.8 1157.02
#Mann= 3 , 0 , 0
       0      .1       0   258.9    .045       0   279.6      .1       0
Bank Sta=258.9,279.6
XS Rating Curve= 0 ,0
Exp/Cntr=0.3,0.1

Type RM Length L Ch R = 1 ,27616.4 ,470.6,464.7,459.3
XS GIS Cut Line= 2
     1835272.168      374552.012     1835444.371      375211.518
#Sta/Elev= 30
       0 1098.66     9.9 1097.44    19.8 1093.82    39.5 1080.73    49.4 1077.31
    59.3 1076.63    69.2 1073.85    88.9 1062.74   118.5 1059.95   128.4 1055.84
   138.3 1047.07   158.1 1035.57   187.7  1024.7   197.6 1021.73   207.4 1020.81
   256.8 1019.25   266.7 1018.57   286.5 1019.22   355.6 1021.48   375.4 1026.64
   434.6 1044.55   444.5 1050.01   474.2  1070.3     484 1074.04   563.1 1075.04
   582.8  1078.1   592.7 1076.33   612.5 1078.29   622.4 1082.54   681.6 1115.16
#Mann= 3 , 0 , 0
       0      .1       0   256.8    .045       0   286.5      .1       0
Bank Sta=256.8,286.5
XS Rating Curve= 0 ,0
Exp/Cntr=0.3,0.1

Type RM Length L Ch R = 1 ,27151.7 ,431.8,435.5,438.4
XS GIS Cut Line= 2
     1834788.333       374733.91     1835135.017      375346.108
#Sta/Elev= 30
       0 1089.37     9.9 1087.26    29.7 1090.52    39.6  1090.9    49.6 1088.91
    69.4  1076.6    89.2  1076.1     109 1072.34   118.9 1067.08   128.8 1063.87
   148.6 1051.66   158.6 1047.57     218  1046.5   237.8 1040.37   297.3 1014.15
   307.2 1013.36   317.1 1014.46   336.9 1025.53   346.8 1027.83   396.4 1027.31
   426.1 1028.84   515.3 1038.28   525.2  1041.5   535.1 1046.96   564.8 1066.58
   574.7  1071.5   594.6 1072.34     654 1071.24   673.8 1078.34   703.6 1095.84
#Mann= 3 , 0 , 0
       0      .1       0   297.3    .045       0   317.1      .1       0
Bank Sta=297.3,317.1
XS Rating Curve= 0 ,0
Exp/Cntr=0.3,0.1

Type RM Length L Ch R = 1 ,26716.3 ,346.1,345.5,345.3
XS GIS Cut Line= 2
     1834422.543      374865.221     1834684.884      375535.761
#Sta/Elev= 30
       0 1084.98    19.7 1085.06    29.6 1088.57    39.4 1087.63    59.2 1079.01
   108.5 1052.98   138.1 1045.62     148 1046.26   157.8 1044.63   187.4 1033.75
     217 1026.79   236.7 1016.69   266.3  1016.7   289.4 1008.84   295.9 1008.04
   319.71011.893   335.4 1013.72   443.9 1011.92   463.6 1013.72   493.2  1025.5
   512.9 1043.07   532.6 1058.79   562.2 1080.03   572.1  1084.4   631.3 1078.21
   680.6 1069.87   690.4  1070.2   700.3  1080.7   710.2 1101.19     720 1118.51
#Mann= 3 , 0 , 0
       0      .1       0   289.4    .045       0   319.7      .1       0
Bank Sta=289.4,319.7
XS Rating Curve= 0 ,0
Exp/Cntr=0.3,0.1

Type RM Length L Ch R = 1 ,26370.8 ,476,472.7,468.7
XS GIS Cut Line= 2
     1834099.261      374990.043     1834382.209      375673.093
#Sta/Elev= 30
       0 1071.34      50 1065.28    69.9 1060.01    99.9 1042.72   109.9 1034.68
   119.9 1029.23   139.9 1025.05   159.9 1017.57   199.8 1012.79   269.8 1010.72
   319.7 1004.74   329.7 1003.76   339.7 1003.96   349.7 1008.49   359.7 1012.35
   379.7 1009.22   419.6 1009.86   439.6 1019.12   469.6 1039.92   509.5 1061.92
   539.5 1066.18   569.5    1081   619.4 1076.21   669.4 1065.01   679.4 1068.79
   689.4 1086.18   699.4 1105.89   709.4 1120.04   729.3 1140.18   739.3  1148.8
#Mann= 3 , 0 , 0
       0     .08       0   319.7    .045       0   349.7      .1       0
Bank Sta=319.7,349.7
XS Rating Curve= 0 ,0
Exp/Cntr=0.3,0.1

Type RM Length L Ch R = 1 ,25898.1 ,424.1,416.7,409.1
XS GIS Cut Line= 2
     1833494.257      374995.981     1834006.017      375825.585
#Sta/Elev= 30
       0 1014.88    89.5 1014.35   109.4 1012.79   119.4 1013.75   139.2 1020.13
   169.1 1020.19     179  1019.6   198.9 1014.37   228.8 1011.08   308.3 1015.36
   328.2 1015.12   348.1 1011.56     368 1010.78   457.5 1010.78   487.4 1014.64
   507.3 1008.72   562.41003.541   576.9 1000.87   606.7  1003.9   676.4 1004.62
   686.3 1007.18   716.1 1026.93   775.8 1060.77   785.8 1066.19   795.7 1068.63
   805.7 1068.48   825.6 1073.22   855.4 1072.14   944.9 1062.25   974.8 1066.93
#Mann= 3 , 0 , 0
       0     .08       0   562.4    .045       0   606.7      .1       0
Bank Sta=562.4,606.7
XS Rating Curve= 0 ,0
Exp/Cntr=0.3,0.1

Type RM Length L Ch R = 1 ,25481.5 ,433.1,407.6,381.9
XS GIS Cut Line= 2
     1833152.194      375483.991     1833725.087      375958.471
#Sta/Elev= 30
       0 1034.24   267.8 1033.04   327.3 1032.22   347.1 1031.34   357.1 1029.76
   376.9 1025.44   426.5 1011.32   446.3 1006.56   456.2 1005.09   466.2 1005.27
     486 1001.92   505.8 1001.96   515.8 1000.38   525.7   997.6   535.6  997.59
   546.7 1002.78   555.4  1007.2   565.3  1010.6   575.3 1013.44   585.2 1016.14
   595.1 1018.06     605 1019.08   614.9 1021.86   634.8 1029.43   674.4 1045.64
   684.4 1049.42   704.2 1051.82   714.1 1055.22     734 1062.79   743.9 1065.52
#Mann= 3 , 0 , 0
       0     .08       0   515.8    .045       0   546.7      .1       0
Bank Sta=515.8,546.7
XS Rating Curve= 0 ,0
Exp/Cntr=0.3,0.1

Type RM Length L Ch R = 1 ,25073.9 ,324.4,324.5,324.5
XS GIS Cut Line= 2
     1833171.889      376280.378     1833746.052      376018.012
#Sta/Elev= 30
       0 1148.05    49.3 1119.78    59.2 1117.09    78.9 1106.72    88.8 1099.36
   118.4  1068.4   128.2 1061.99   157.8  1054.3   197.3 1055.64   207.1 1053.39
   236.7 1034.52   256.4  1018.5   266.3 1016.72   276.2 1011.83     286 1004.24
   295.9  999.11   305.8  996.17   315.6  995.54   325.5  995.71   335.4  998.86
   355.1 1004.29   394.5    1019   424.1 1021.55   453.7  1031.6   473.4 1039.87
     503 1048.59   532.6 1052.47   601.7 1074.03   611.5 1075.42   631.3 1075.43
#Mann= 3 , 0 , 0
       0      .1       0   295.9    .045       0   335.4      .1       0
Bank Sta=295.9,335.4
XS Rating Curve= 0 ,0
Exp/Cntr=0.3,0.1

Type RM Length L Ch R = 1 ,24749.4 ,398.9,404.3,409.9
XS GIS Cut Line= 2
     1833273.508      376584.476     1833852.372      376319.962
#Sta/Elev= 30
       0 1098.99    49.7 1089.63    59.7 1087.13    79.6 1079.64    89.5  1073.5
   109.4 1054.47   119.3 1049.35   149.2  1048.8     169 1051.34   188.9 1049.46
   238.7 1051.23   248.6 1049.42   288.4 1024.13   328.2 1007.82   338.1 1006.12
     358 1005.92   367.9 1003.75   377.9  999.25   397.8  995.11   417.2  994.45
   433.8997.0226   457.4 1005.36   487.3 1018.68   507.2 1023.16   546.9 1041.74
   566.8 1049.53   586.7 1053.85   596.7 1058.08   616.6  1063.8   636.4 1065.82
#Mann= 3 , 0 , 0
       0      .1       0   397.8    .045       0   433.8      .1       0
Bank Sta=397.8,433.8
XS Rating Curve= 0 ,0
Exp/Cntr=0.3,0.1

Type RM Length L Ch R = 1 ,24345.1 ,633.3,664.1,692.2
XS GIS Cut Line= 2
     1833217.974      376887.009     1833997.152      376744.227
#Sta/Elev= 30
       0  1045.1    59.4 1037.04   108.9 1038.72   128.7 1037.33   188.1 1029.79
   237.6 1026.22   247.6 1024.55   287.2 1015.25   316.9 1010.47   445.6 1004.55
   455.5 1003.45   465.4 1000.68   475.3 1001.06   485.2 1000.08   495.1  994.17
     505  992.16   508.9992.1405   514.9  992.12   537.2995.6493   554.5 1001.36
   594.1 1018.25     604 1021.26   623.8 1025.09   653.5 1037.14   663.4 1040.11
   673.3 1040.95   722.8 1040.54   752.5  1037.7   782.2 1038.33   792.2 1039.78
#Mann= 3 , 0 , 0
       0      .1       0   508.9    .045       0   537.2      .1       0
Bank Sta=508.9,537.2
XS Rating Curve= 0 ,0
Exp/Cntr=0.3,0.1

Type RM Length L Ch R = 1 ,23681   ,91.7,80.1,70.8
XS GIS Cut Line= 4
     1833510.708      377612.073     1833898.957      377360.699
     1833999.213      377454.844     1834188.252      377445.907
#Sta/Elev= 30
       0  999.03   108.2  999.05     187  997.64   226.3  998.28   314.9  997.15
   354.3  995.62   442.8  993.28   462.5  992.37   482.2  992.08   501.8  991.51
   511.6  991.08   528.5989.0786   541.1  987.79   550.9  987.57   560.8   988.5
   565.3989.4459   570.6  990.56   580.4  992.05   590.2  992.99     600  993.04
     610  994.31   629.9  996.32   649.8 1000.89   659.8 1001.79   689.7 1002.79
   719.6 1004.81   749.5 1006.27   759.4 1007.07   779.3 1009.14   789.3  1009.7
#Mann= 3 , 0 , 0
       0     .06       0   528.5    .045       0   565.3     .06       0
Bank Sta=528.5,565.3
XS Rating Curve= 0 ,0
Exp/Cntr=0.3,0.1

Type RM Length L Ch R = 1 ,23600.9 ,348.5,337.7,326.5
XS GIS Cut Line= 5
     1833610.879       377620.42     1833876.331      377442.357
     1833982.401      377518.157     1834452.423       377446.59
     1834994.012      377276.377
#Sta/Elev= 30
       0  999.08   129.8  999.12   289.7   995.6   356.9  995.95   366.2  995.27
     381991.3212   394.1   987.4   403.4  987.32   422.1  990.27   431.4  992.47
   479.7  994.79   539.2  994.53   598.6 1007.91   618.4 1007.45   648.1  1013.2
   677.8 1015.42   697.6 1013.27   727.4 1013.97   737.3 1012.79   757.1 1005.63
   776.9 1003.28   816.5  1003.7     866 1012.84   915.6 1000.58   925.4  999.54
  1064.9 1001.86  1244.2  999.81  1333.8 1000.71  1433.4 1017.33  1493.2 1017.88
#Mann= 3 , 0 , 0
       0     .06       0     381    .045       0   422.1     .06       0
Bank Sta=381,422.1
XS Rating Curve= 0 ,0
Exp/Cntr=0.3,0.1

Type RM Length L Ch R = 1 ,23263.2 ,294.2,300,306
XS GIS Cut Line= 2
     1833419.189      377730.584     1835274.651      378025.933
#Sta/Elev= 30
       0  1018.4      60 1018.71   109.9 1016.25   119.9    1015   159.9 1000.11
   219.9 1001.07   239.8  998.33   519.7  999.05   529.7  998.86   549.2992.8645
   569.6  985.53   589.6  985.06   611.5987.2333   649.6  996.52   789.5 1001.18
   809.5 1004.69   939.4 1014.08   949.4 1018.82   999.4 1051.56  1059.3 1072.46
  1149.3 1091.94  1199.2 1106.71  1279.2 1126.82  1409.1 1153.81  1479.1 1164.07
    1549 1168.75    1639 1169.58  1698.9 1167.74  1738.9 1164.18  1878.8  1140.9
#Mann= 3 , 0 , 0
       0     .08       0   549.2    .045       0   611.5     .08       0
Bank Sta=549.2,611.5
XS Rating Curve= 0 ,0
Exp/Cntr=0.3,0.1

Type RM Length L Ch R = 1 ,22963.2 ,394.8,394.1,393.3
XS GIS Cut Line= 2
     1833368.011      377871.527     1834372.245      378300.455
#Sta/Elev= 30
       0 1084.89   109.2 1063.84   178.7 1035.75   238.2 1015.53     268 1015.32
     278 1013.14   307.8 1000.44   317.7  997.81     407  1000.5   486.4   998.5
   515.2988.0115   536.1  985.11   555.9  986.18   566.9990.2043   595.6 1000.16
   665.1 1003.43   734.6  1003.1   754.5 1005.91   784.2 1015.33     814  1015.9
     824 1020.24   843.8 1032.46   873.6 1044.01   913.3 1051.18   933.2  1062.3
     953 1069.32  1012.6 1083.44  1042.4 1088.66  1072.2 1103.12    1092 1108.48
#Mann= 3 , 0 , 0
       0     .08       0   515.2    .045       0   566.9     .06       0
Bank Sta=515.2,566.9
XS Rating Curve= 0 ,0
Exp/Cntr=0.3,0.1

Type RM Length L Ch R = 1 ,22569.1 ,705.7,714.8,723.9
XS GIS Cut Line= 2
     1833394.882      378322.471     1834115.283      378598.361
#Sta/Elev= 30
       0 1047.68    49.4 1027.67      89 1015.01    98.9 1010.47   108.8 1007.23
   148.4  1005.1   187.9 1004.47   207.7  1006.1   227.5 1010.55   247.2 1010.54
   257.1 1008.45   276.9 1001.22   296.7  998.31   306.6  995.57   329.2 984.736
   336.3   982.4   344.4  982.39     356   982.7   365.9  984.21   405.5  984.26
   415.4  985.18     445  993.89   454.9  994.28   553.8  995.01     633  994.45
   642.8  996.56   652.7 1000.11   672.5 1001.36   702.2 1007.89   771.4 1019.03
#Mann= 3 , 0 , 0
       0     .08       0   329.2    .045       0   365.9     .06       0
Bank Sta=329.2,365.9
XS Rating Curve= 0 ,0
Exp/Cntr=0.3,0.1

Type RM Length L Ch R = 1 ,21854.3 ,811.8,795.8,778.5
XS GIS Cut Line= 4
     1832813.417      378522.736     1833299.999      378987.609
     1833424.713      379014.021     1834013.255      378685.896
#Sta/Elev= 30
       0 1144.46    19.8 1138.51    49.5 1123.64      99 1104.51   118.8  1099.7
   197.9 1067.78   217.7 1062.65   267.2 1044.59   296.9 1040.64   336.5  1046.2
   366.2  1046.4   425.6 1026.38   445.3 1022.49   494.8  998.96   524.5  993.49
   556.4  981.17     574  979.94     596982.2789   623.5  989.71   731.8  992.87
   889.6   991.4  1107.6   993.6  1256.3  992.52  1295.9   989.6  1365.3  991.61
  1385.1  998.73  1414.8 1003.92  1454.4 1003.28  1464.4  999.74  1474.3  999.32
#Mann= 3 , 0 , 0
       0     .08       0   556.4    .045       0     596     .06       0
Bank Sta=556.4,596
XS Rating Curve= 0 ,0
Exp/Cntr=0.3,0.1

Type RM Length L Ch R = 1 ,21058.5 ,380,389.2,399
XS GIS Cut Line= 2
     1832509.757      379554.042      1833806.63      379590.125
#Sta/Elev= 30
       0 1127.61      20  1123.9    39.9 1122.84    89.8 1110.61   149.7 1088.34
   219.6 1067.74   249.5 1056.23   309.4 1041.68   349.3 1027.27   409.2  986.16
   419.2  981.45   431.6977.9874   449.1  977.73   467.9979.5978     479  981.61
   618.8  981.77   688.6  983.91   718.6  986.99   748.5  995.48   758.5  995.58
   828.3 1017.23   878.2 1039.79   938.1 1058.85   948.1 1061.76    1008 1071.73
  1087.8 1094.75  1097.8  1098.1  1177.6 1134.43  1217.5 1145.52  1297.4 1158.25
#Mann= 3 , 0 , 0
       0      .1       0   431.6    .045       0   467.9     .06       0
Bank Sta=431.6,467.9
XS Rating Curve= 0 ,0
Exp/Cntr=0.3,0.1

Type RM Length L Ch R = 1 ,20669.3 ,136.4,137.8,139.2
XS GIS Cut Line= 3
      1832682.32      379777.714     1833098.659      379983.284
     1833817.859       380098.73
#Sta/Elev= 30
       0 1032.08    39.5 1025.22    49.4 1021.98      79 1008.55    88.9 1007.48
   118.6 1011.07   148.2 1010.12   217.3  994.31   256.9  989.08   286.5  981.07
   345.8  979.43   366.1  976.57   375.4  976.26   395.2  976.42   400.2977.8384
   414.9  981.21   444.6  983.68   524.2  985.56   554.1  987.65   584.1  987.75
     624  991.95   663.9  993.52   743.7 1019.55   883.4 1049.04   923.3 1053.51
   973.2 1054.44  1013.1 1056.91  1043.1 1056.14    1083 1058.93  1192.7 1075.27
#Mann= 3 , 0 , 0
       0      .1       0   366.1    .045       0   400.2     .06       0
Bank Sta=366.1,400.2
XS Rating Curve= 0 ,0
Exp/Cntr=0.3,0.1

Type RM Length L Ch R = 1 ,20531.5 ,623.1,614.5,605.1
XS GIS Cut Line= 3
      1832635.39      379881.759     1833051.081      380119.698
     1833734.526      380230.674
#Sta/Elev= 30
       0 1029.24    29.9 1033.07    59.9 1047.07    79.8 1045.95   119.7  1036.2
   139.7 1028.75   199.6 1004.93   239.5  982.48   249.5  979.28   309.3  980.18
   329.3  977.36   359.2  976.04   379.2  977.95   419.1  978.94     469  984.46
   548.2  985.86   637.2     993   686.7  994.02   706.5  990.96   736.2  993.92
   785.6  996.04   815.3  995.46   894.4 1002.98   914.2 1003.08     934 1000.92
  1003.2 1006.82  1072.4 1009.36  1092.2  1007.6  1121.9 1010.99  1171.4 1013.59
#Mann= 3 , 0 , 0
       0      .1       0   329.3    .045       0   379.2     .06       0
Bank Sta=329.3,379.2
XS Rating Curve= 0 ,0
Exp/Cntr=0.3,0.1

Type RM Length L Ch R = 1 ,19917   ,338,337.2,336.4
XS GIS Cut Line= 2
     1832316.412      380431.219     1833410.992      380600.666
#Sta/Elev= 30
       0 1133.01    39.9 1130.08    69.8 1125.17    89.8 1121.15   109.8 1113.67
   229.5 1054.16   279.4 1033.81   299.4 1019.32   339.3  981.42   352.7 974.047
   359.2  972.52     394973.8536   419.1  975.97   548.8  979.74   648.6  979.02
   678.5  980.43   688.5   982.8   718.5  994.77   738.4 1005.22   798.3 1022.88
   818.2 1026.62   828.2 1026.44   848.2 1034.89   888.1 1045.89     928 1051.17
     948 1056.91   997.8 1066.27  1027.8 1077.11  1077.7 1099.58  1107.6 1108.88
#Mann= 3 , 0 , 0
       0      .1       0   352.7    .045       0     394     .08       0
Bank Sta=352.7,394
XS Rating Curve= 0 ,0
Exp/Cntr=0.3,0.1

Type RM Length L Ch R = 1 ,19579.9 ,514.2,513.1,512.1
XS GIS Cut Line= 2
     1832211.917       380768.14     1833297.526      380898.626
#Sta/Elev= 30
       0 1103.23    39.8 1099.96    89.5    1094   129.2 1086.88   218.7 1059.54
   288.3 1040.96   347.9 1027.44   377.7 1018.54   397.6 1010.27   427.4  991.71
   447.3  976.13   457.2     971     497  970.32     507  971.77   516.9  974.16
   576.5  975.53   616.3   978.4   705.8  976.43   735.6  976.91   755.5  982.31
   775.3  991.98   795.2 1004.58   815.1 1015.11   844.9  1025.4   914.5 1041.83
   944.3 1044.93  1023.8 1066.73  1053.7 1071.14  1063.6 1076.78  1093.4 1087.71
#Mann= 3 , 0 , 0
       0      .1       0   457.2    .045       0     507     .08       0
Bank Sta=457.2,507
XS Rating Curve= 0 ,0
Exp/Cntr=0.3,0.1

Type RM Length L Ch R = 1 ,19066.7 ,796.8,783.7,769.5
XS GIS Cut Line= 2
     1832088.014      381279.152     1833191.562       381362.23
#Sta/Elev= 30
       0 1033.18      10 1028.09    29.9 1020.75    39.9 1016.13    49.8 1015.12
    79.8  1017.7   119.6 1025.54   129.6 1026.27   189.4 1025.97   239.3 1023.31
   309.1 1014.06   398.8   998.4   468.6  984.53   528.4  975.48   618.1  972.05
   628.1  970.24   638.1  968.07     658  967.43   669.2970.2408     678  971.86
   737.8  973.85   817.5  973.69   827.5   975.6   837.5  978.82   867.4  991.62
   887.3   998.3   967.1 1015.47  1036.9 1037.88  1066.8 1040.86  1106.7 1052.43
#Mann= 3 , 0 , 0
       0      .1       0   628.1    .045       0   669.2     .08       0
Bank Sta=628.1,669.2
XS Rating Curve= 0 ,0
Exp/Cntr=0.3,0.1

Type RM Length L Ch R = 1 ,18283.1 ,360,366.6,373
XS GIS Cut Line= 2
     1832249.828       382316.83     1833192.899      381761.134
#Sta/Elev= 30
       0 1100.32    79.6 1093.74   228.9 1084.17   258.7 1079.64   278.6 1073.51
   298.5  1065.4   318.4 1055.96   348.3 1039.22   358.2  1035.2   378.1 1028.67
   417.9  1007.5   487.6  975.96   507.5  965.84   510.1965.5415   525.2  964.68
   537.5965.3629   547.3   967.6   557.3   968.6   646.8  970.24   666.7  973.11
   686.6  977.34   696.6  978.26   736.4  979.29   786.1   984.6   835.9  986.16
   945.4  999.74   975.2 1005.65  1054.8 1016.51  1074.7 1017.36  1094.6 1023.63
#Mann= 3 , 0 , 0
       0      .1       0   510.1    .045       0   537.5     .08       0
Bank Sta=510.1,537.5
XS Rating Curve= 0 ,0
Exp/Cntr=0.3,0.1

Type RM Length L Ch R = 1 ,17916.5 ,839.4,866.9,892.9
XS GIS Cut Line= 2
     1832523.556       382454.42     1833615.742      382180.787
#Sta/Elev= 30
       0 1077.42    49.8  1064.4    79.7 1059.29   129.5 1057.12   149.5 1054.18
   179.4 1046.59   209.2 1036.82   239.1 1031.06     269 1022.62     279 1019.21
     289 1013.12   298.9 1005.34   318.8  987.05   328.8   979.5   358.7  965.88
   374.6963.0218   398.6  962.76   408.8963.0113   438.4  970.46   597.8  975.51
   647.7  978.23   687.5  981.94   697.5  985.23   707.4  991.01   727.4  997.63
     847 1020.35   936.6 1047.03  1036.3 1074.47  1086.1 1091.53  1125.9 1098.19
#Mann= 3 , 0 , 0
       0      .1       0   374.6    .045       0   408.8     .08       0
Bank Sta=374.6,408.8
XS Rating Curve= 0 ,0
Exp/Cntr=0.3,0.1

Type RM Length L Ch R = 1 ,17049.6 ,227.7,224.6,222.7
XS GIS Cut Line= 2
     1832451.425      382515.048     1833149.878      383484.602
#Sta/Elev= 30
       0 1075.47      10 1075.11    19.9 1072.31    49.8 1061.41   109.5  1036.2
   139.4 1025.09   159.3 1015.86   179.2 1009.51   209.1  995.82   248.9   982.2
   268.9  977.53   298.7  973.74   378.4   970.3   557.6  967.93   597.5  961.78
   617.4  959.66   637.3  959.71   647.8961.4926   677.1  965.06     697  973.27
     717  977.16   736.9 1001.54   746.8 1011.84   756.8 1018.84   876.3 1071.23
   916.1 1084.34     956 1091.02  1045.6 1098.92  1115.3 1100.77  1194.9 1098.87
#Mann= 3 , 0 , 0
       0      .1       0   597.5    .045       0   647.8      .1       0
Bank Sta=597.5,647.8
XS Rating Curve= 0 ,0
Exp/Cntr=0.3,0.1

Type RM Length L Ch R = 1 ,16825   ,372.7,365.1,361.5
XS GIS Cut Line= 2
     1832247.214      382730.669       1833021.5      383553.848
#Sta/Elev= 30
       0 1070.14    49.6 1045.67   128.9 1016.46   188.4  983.35   218.1  971.98
     228  970.26   356.9  968.45   416.4   965.3   465.9  964.96   515.5  971.29
   525.4  970.66   560.9961.2761     575  958.16   594.8  957.88   600.8959.4497
   614.6  962.16   634.4  962.65   644.4  966.56   664.2  977.74     684  980.54
   693.9   989.9   703.8  1002.2   713.8 1009.86   783.1 1036.34   852.5 1069.46
   882.3 1080.35   902.1 1085.74   931.8 1090.16   961.6 1090.85  1130.1 1077.86
#Mann= 3 , 0 , 0
       0      .1       0   560.9    .045       0   600.8      .1       0
Bank Sta=560.9,600.8
XS Rating Curve= 0 ,0
Exp/Cntr=0.3,0.1

Type RM Length L Ch R = 1 ,16459.9 ,648.3,639.7,627.1
XS GIS Cut Line= 2
     1831874.865      382939.337       1832809.3      383735.504
#Sta/Elev= 30
       0 1115.32    79.8 1099.69   109.8 1092.34   139.7 1078.51   209.6 1042.72
   219.6 1038.37   279.5 1014.76   299.4 1007.89   329.4  999.46   389.2  974.98
   409.2  969.26   479.1  962.91   588.9  960.41   608.8  957.92   628.8  956.75
   638.8  956.75   648.7   959.7   658.7  962.56   728.6  967.65   748.6  970.53
   768.5  971.55   778.5  973.76   788.5  978.42   848.4 1000.49   888.3 1017.14
   938.2 1030.36   968.1 1036.27   988.1 1038.22    1008 1038.17  1227.6 1026.87
#Mann= 3 , 0 , 0
       0      .1       0   608.8    .045       0   648.7      .1       0
Bank Sta=608.8,648.7
XS Rating Curve= 0 ,0
Exp/Cntr=0.3,0.1
